--- POCARN.prj (project) ---

Proj Title=POCARN
Current Plan=p01
Default Exp/Contr=0,0
English Units
Geom File=g01
Flow File=f01
Plan File=p01
Background Map Layer=Inundation Boundary (01pct Value_0)
Background Map Layer=Inundation Boundary (01pct Value_0)
BEGIN DESCRIPTION:
----------MODEL BY WOOD PLC 2021----------
Stream Name: Poca Run
Flood Zone: Enhanced Approximate
Pocahontas County, WV
HEC-RAS Version: RAS 6.1
Vertical Datum: NAVD88
Projection: NAD 1983 StatePlane West Virginia S FIPS 4702 (US Feet)
Terrain: 1-meter LIDAR (FEMA Region III 3DEP collected 2016-2018)
Land Use: 2019 NLCD
Hydrologic Method:
WV SIR2010-5033 regression equations
Model Notes:
Normal depth tie in with Eastfork Greenbrier river
END DESCRIPTION:
DSS Export Rating Curves= 0
DSS Export Rating Curve Sorted= 0
DSS Export Volume Flow Curves= 0
DXF OffsetX= 0
DXF OffsetY= 0
DXF ScaleX= 0
DXF ScaleY= 0

--- POCARN.p01 (plan) ---

Plan Title=Floodplain
Program Version=6.10
Short Identifier=Floodplain
Geom File=g01
Flow File=f01
Subcritical Flow
K Sum by GR= 0
Std Step Tol= 0.01
Critical Tol= 0.01
Num of Std Step Trials= 20
Max Error Tol= 0.3
Flow Tol Ratio= 0.001
Split Flow NTrial= 30
Split Flow Tol= 0.02
Split Flow Ratio= 0.02
Log Output Level= 0
Friction Slope Method= 1
Unsteady Friction Slope Method= 2
Unsteady Bridges Friction Slope Method= 1
Parabolic Critical Depth
Global Vel Dist= 0 , 0 , 0
Global Log Level= 0
CheckData=True
Encroach Param=-1 ,0,0, 0
Mapping Interval=1HOUR
Computation Time Step Use Courant=        0
Computation Time Step Use Time Series=    0
Computation Time Step Count To Double=0
Computation Time Step Max Doubling=0
Computation Time Step Max Halving=0
Computation Time Step Residence Courant=0
Run HTab= 0
Run UNet= 0
Run Sediment= 0
Run PostProcess= 0
Run WQNet= 0
Run RASMapper=-1
UNET Theta= 0
UNET Theta Warmup= 0
UNET ZTol= 0
UNET ZSATol= 0
UNET MxIter= 0
UNET Max Iter WO Improvement= 0
UNET MaxInSteps= 0
UNET DtIC= 0
UNET DtMin= 0
UNET MaxCRTS= 0
UNET WFStab= 0
UNET SFStab= 0
UNET WFX= 1
UNET SFX= 1
UNET Gravity=32.174
UNET 1D Methodology=Finite Difference
UNET DSS MLevel= 1
UNET Pardiso=0
UNET DZMax Abort= 0
UNET Use Existing IB Tables= 0
UNET Froude Reduction=False
UNET Froude Limit= 0
UNET Froude Power= 0
UNET D1 Cores= 0
UNET WindReference=Eulerian
UNET WindDragFormulation=Hsu (1988)
UNET D2 Coriolis=0
UNET D2 Cores= 0
UNET D2 Theta= 1
UNET D2 Theta Warmup= 1
UNET D2 Z Tol= 0.01
UNET D2 Volume Tol= 0.01
UNET D2 Max Iterations= 20
UNET D2 Equation= 0
UNET D2 RampUpFraction=0.1
UNET D2 TimeSlices= 1
UNET D2 Turbulence Formulation=Non-Conservative (original)
UNET D2 Eddy Viscosity=0.3
UNET D2 Transverse Eddy Viscosity=0.1
UNET D2 Smagorinsky Mixing=0
UNET D2 BCVolumeCheck=0
UNET D2 Cores=0
UNET D2 SolverType=PARDISO (Direct)
UNET D2 Minimum Iterations= 2147483647
UNET D2 Maximum Iterations= 2147483647
UNET D2 Restart Number= 10
UNET D2 Relaxation Coeff=1.3
UNET D2 SOR Precondition Iterations= 10
UNET D2 ILUT Maximum Fill= 8
UNET D2 ILUT Tolerance=1E-08
UNET D1D2 MaxIter= 0
UNET D1D2 ZTol=0.01
UNET D1D2 QTol=0.1
UNET D1D2 MinQTol=1
Write IC File= 0
Write IC File at Fixed DateTime=0
Write IC File at Sim End=0
Echo Input=False
Echo Parameters=False
Echo Output=False
Write Detailed= 0
HDF Write Warmup=0
HDF Write Time Slices=0
HDF Flush=0
HDF Compression= 1
HDF Chunk Size= 1
HDF Spatial Parts= 1
HDF Use Max Rows=0
HDF Fixed Rows= 1
Calibration Method= 0
Calibration Iterations= 20
Calibration Max Change=0.05
Calibration Tolerance=0.2
Calibration Maximum=1.5
Calibration Minimum=0.5
Calibration Optimization Method= 1
WQ AD Non Conservative
WQ ULTIMATE=-1
WQ Max Comp Step=1HOUR
WQ Output Interval=15MIN
WQ Output Selected Increments= 0
WQ Output face flow=0
WQ Output face velocity=0
WQ Output face area=0
WQ Output face dispersion=0
WQ Output cell volume=0
WQ Output cell surface area=0
WQ Output cell continuity=0
WQ Output cumulative cell continuity=0
WQ Output face conc=0
WQ Output face dconc_dx=0
WQ Output face courant=0
WQ Output face peclet=0
WQ Output face adv mass=0
WQ Output face disp mass=0
WQ Output cell mass=0
WQ Output cell source sink temp=0
WQ Output nsm pathways=0
WQ Output nsm derived pathways=0
WQ Create Restart=0
WQ Fixed Restart=0
WQ System Summary=0
WQ Write To DSS=0
Sorting and Armoring Iterations= 10
XS Update Threshold= 0.02
Bed Roughness Predictor= 0
Hydraulics Update Threshold= 0.02
Energy Slope Method= 1
Volume Change Method= 1
Sediment Retention Method= 0
Sediment TS Multiplier= 1
Warm Up Method= 0
XS Weighting Method= 0
Number of US Weighted Cross Sections= 1
Number of DS Weighted Cross Sections= 1
Upstream XS Weight=0
Main XS Weight=1
Downstream XS Weight=0
Number of DS XS's Weighted with US Boundary= 1
Upstream Boundary Weight= 1
Weight of XSs Associated with US Boundary= 0
Number of US XS's Weighted with DS Boundary= 1
Downstream Boundary Weight= 0.5
Weight of XSs Associated with DS Boundary= 0.5
Percentile Method= 0
Sediment Output Level= 3
Mass or Volume Output= 0
Output Increment Type= 1
Profile and TS Output Increment= 1
Transport Output Increment 1
XS Output Flag= 0
XS Output Increment= 10
Read HDF5 Sediment Hotstart= 0
Sediment Hotstart Type= 0
Write Gradation File= 0
Read Gradation Hotstart= 0
Write HDF5 File= 1
Write Binary Output= 1
Write DSS Sediment File= 0
DSS Sediment Output Type= 1
SV Curve= 0
Specific Gage Flag= 0
Subcell Erosion Methods= 0
Subcell Deposition Methods= 0
Advection Scheme= 1
Matrix Solver= 0
Implicit Weighting Factor= 1
Maximum Outer Loop Convergence Iterations= 5
Convergence Maximum Absolute= 0.001
Convergence RMSE= 0.0001
Grain Fractions Max Abs Error= 0.001
Max Subgrid Regions= 1
Max Subgrid Length Scale= 3.402823E+38
Initial Layer Thickness= 3.402823E+38
Min Layer Thickness= 3.402823E+38
Max Layer Thickness= 3.402823E+38
Number of Layers= 5

--- POCARN.f01 (steady flow) ---

Flow Title=Flow
Program Version=6.10
Number of Profiles= 6
Profile Names=01pct,10pct,04pct,02pct,0_2pct,01plus
River Rch & RM=POCARN,Main            ,9848
     860     462     609     731    1190    1270
River Rch & RM=POCARN,Main            ,3476
    1090     588     772     924    1500    1610
River Rch & RM=POCARN,Main            ,1466
    1480     809    1060    1260    2030    2180
Boundary for River Rch & Prof#=POCARN,Main            , 1
Up Type= 0
Dn Type= 3
Dn Slope=0.01532
Boundary for River Rch & Prof#=POCARN,Main            , 2
Up Type= 0
Dn Type= 3
Dn Slope=0.01532
Boundary for River Rch & Prof#=POCARN,Main            , 3
Up Type= 0
Dn Type= 3
Dn Slope=0.01532
Boundary for River Rch & Prof#=POCARN,Main            , 4
Up Type= 0
Dn Type= 3
Dn Slope=0.01532
Boundary for River Rch & Prof#=POCARN,Main            , 5
Up Type= 0
Dn Type= 3
Dn Slope=0.01532
Boundary for River Rch & Prof#=POCARN,Main            , 6
Up Type= 0
Dn Type= 3
Dn Slope=0.01532
DSS Import GetInterval= 0
DSS Import GetPeak= 0
DSS Import FillOption= 0

--- POCARN.g01 (geometry) ---

Geom Title=Geometry
Program Version=6.10

River Reach=POCARN          ,Main
Reach XY= 30
2343935.26085855580645.0507138972343550.24705345580467.142559247
2343497.85273296580311.5776700522343233.81442221580254.713213669
2342846.16625197 579821.473948972342729.45861372579508.556964666
2342430.97023197579348.1235177222342267.47024339578935.440413348
 2342337.3585642578588.9831388942342241.71043989578298.060657233
2342292.69524606577743.5893252342342515.33104566577347.511753862
 2342361.0093923577048.9200490962342029.15176084576875.940364033
2341834.17847045 576635.319442482341670.78244789576624.471812814
 2341539.4773269576452.8473909792341301.28983711576424.590564107
2341134.27325058576292.9870459532340781.79655586576288.038910683
2340339.53979536576338.7496245152340102.73587901576489.168891232
2339907.61654718576474.0914883182339552.37612256576589.731660274
2339423.51214603576660.0116040162339416.89790106576745.884239517
2339271.50592828576765.1096243472338878.41308515577210.151466411
2338782.28616101 577557.276470282338451.31158015577672.435907369

Type RM Length L Ch R = 1 ,9848    ,306.4,306.4,306.4
XS GIS Cut Line= 4
2344031.32963028580586.5258037692343986.46685597580623.565736442
2343893.49036082580644.909740491 2343801.2727836580766.493447555
#Sta/Elev= 30
       0 3294.81     9.8 3292.28    24.8 3290.27    48.1 3285.75      56 3281.81
    72.8 3271.33    76.9 3269.94    81.5  3269.3    89.3    3270    93.4 3269.69
100.52753267.822   105.7 3267.59     119 3267.77   126.2 3268.67   141.5 3268.61
   153.9  3271.4   158.9 3269.77   166.1 3269.22     169 3269.69   174.7 3272.47
     179 3273.83   189.1 3274.63   200.4 3274.09   214.2 3277.84   229.2 3279.25
   257.5 3280.83   280.3 3280.77   284.4 3281.32   297.5 3286.93   306.2    3288
#Mann= 4 ,-1,0
       0      .1       0100.5275    .045       0     119      .1       0
  233.57     .06       0
Bank Sta=100.5275,119
XS Rating Curve= 0 ,0
Exp/Cntr=0.3,0.1

Type RM Length L Ch R = 1 ,9541    ,167.5,168.9,168.8
XS GIS Cut Line= 3
2343768.24379138580423.3141792782343655.15436969580560.211900282
2343594.26006569580679.711248717
#Sta/Elev= 30
       0 3285.08    31.5 3273.46    46.8 3269.58    59.5 3267.22    80.2 3265.64
    92.3 3265.41   106.2 3262.51   109.3 3261.25     115 3256.32   117.9  3254.8
   125.7 3253.93   132.7 3254.79   140.6 3256.32   154.8  3257.2   168.4 3256.68
   180.5 3258.01   192.4 3256.78   210.6 3256.14   219.1  3254.3   225.1  3254.3
   228.1 3255.08   232.5 3257.94   241.5 3266.97   245.9 3270.13   251.9 3272.66
   257.8 3274.05   290.9 3277.13   296.5 3281.29   305.4 3291.19   311.7 3296.83
#Mann= 4 ,-1,0
       0      .1       0   117.9    .045       0   132.7      .1       0
  197.57     .06       0
Bank Sta=117.9,132.7
XS Rating Curve= 0 ,0
Exp/Cntr(USF)=0,0
Exp/Cntr=0.3,0.1

Type RM Length L Ch R = 1 ,9372    ,371.2,369,364.4
XS GIS Cut Line= 2
2343642.88393851 580349.416881052343423.66444414580570.284642296
#Sta/Elev= 30
       0 3286.93     9.5 3281.31    15.2 3278.89    27.8 3271.63      56 3257.53
    67.3 3252.45    78.6 3250.24    86.6 3249.24    94.7 3248.92   106.4 3249.26
   111.7 3248.37   117.7 3246.66   128.8 3247.76   137.5 3247.37   143.2 3246.43
   146.2 3245.99   154.5 3246.36   171.5 3248.03   182.8    3248   191.2 3248.81
   208.3 3249.45   213.9 3252.44   230.7 3264.41   236.5 3266.87   239.3 3266.53
   247.8 3263.86   284.6 3266.84   293.1  3266.1   298.4 3268.35311.1909 3278.53
#Mann= 5 ,-1,0
       0      .1       0     130     .06       0   143.2    .045       0
   154.5     .06       0     270      .1       0
#XS Ineff= 2 , 0
                          176.16         3255.49
Permanent Ineff=
       F       F
Bank Sta=143.2,154.5
XS Rating Curve= 0 ,0
Exp/Cntr(USF)=0,0
Exp/Cntr=0.3,0.1

Type RM Length L Ch R = 1 ,9003    ,201.3,207,211.7
XS GIS Cut Line= 3
2343340.01490023580206.4297296472343267.49115773580350.241014488
2343227.93275273580400.101087456
#Sta/Elev= 30
       0 3284.21    16.5 3273.29    22.8 3268.53    34.4 3257.87    43.4 3250.84
    52.9 3241.26    56.8 3238.09    61.3 3235.62    70.4 3232.45    83.7 3231.12
    92.7 3230.19   100.2 3230.54   103.2 3231.33   106.2 3232.92   110.6 3234.62
   118.1 3235.02   119.6 3235.44     124 3238.22     133 3242.01   137.5 3244.33
   142.1 3246.08   146.4 3247.11   160.2 3249.36   179.3 3250.16   185.7 3250.23
   192.1 3249.74   195.4 3250.71   205.4 3256.12   216.8 3260.13224.7099 3261.86
#Mann= 5 ,-1,0
       0      .1       0    83.7    .045       0   103.2      .1       0
     140     .06       0  181.06      .1       0
Bank Sta=83.7,103.2
XS Rating Curve= 0 ,0
Exp/Cntr(USF)=0,0
Exp/Cntr=0.3,0.1

Type RM Length L Ch R = 1 ,8796    ,239.5,240.4,241.1
XS GIS Cut Line= 2
2343208.56561695580098.4682493372343044.97512961 580244.75193449
#Sta/Elev= 30
       0 3281.08     4.1 3278.38    13.5 3270.18    19.2 3265.76    24.9 3262.41
    43.5 3253.27    46.1 3251.43    52.1 3246.32    64.5 3232.88    70.2 3227.82
    75.6 3225.83    81.5 3225.64    86.4 3223.89    94.1 3222.74    98.5 3223.01
   101.3 3223.78   104.2 3225.75   107.8 3229.41   112.1 3232.62   118.3 3234.72
   145.4 3235.74   156.1 3234.72   163.7  3235.8   184.1 3236.97   189.2 3238.08
   194.8 3240.84   200.5 3242.91     209 3244.52   215.2 3247.58219.4556 3248.26
#Mann= 5 ,-1,0
       0      .1       0      70     .06       0    86.4    .045       0
   101.3     .06       0     200      .1       0
Bank Sta=86.4,101.3
XS Rating Curve= 0 ,0
Exp/Cntr(USF)=0,0
Exp/Cntr=0.3,0.1

Type RM Length L Ch R = 1 ,8556    ,212.5,218.9,222.2
XS GIS Cut Line= 2
2343035.08552836 579936.938095592342903.63624508580041.190975432
#Sta/Elev= 30
       0  3250.3     3.7 3247.85     8.8 3243.34    13.9 3239.23      19 3235.71
    27.9 3231.89    34.3 3227.94      39 3225.72      45 3224.49    47.8 3223.34
    49.7 3222.23    54.8 3218.41   57.79    3217    59.9 3216.41    67.7 3216.32
    76.3 3216.94    80.3 3217.14    90.5 3221.25    96.2 3222.19   110.4 3222.46
   122.7 3222.34   126.2 3222.07   131.3 3221.09   136.1 3221.18   141.6 3223.51
   150.3 3227.94   156.9 3230.16   161.7 3232.14   164.5 3232.79167.7724 3232.99
#Mann= 4 ,-1,0
       0     .06       0   57.79    .045       0    76.3     .06       0
     160      .1       0
Bank Sta=57.79,76.3
XS Rating Curve= 0 ,0
Exp/Cntr(USF)=0,0
Exp/Cntr=0.3,0.1

Type RM Length L Ch R = 1 ,8337    ,266.4,266.3,264.5
XS GIS Cut Line= 4
2342944.51756392579753.5396972732342869.22636099579802.885958653
 2342799.0224015579826.7960028272342716.10033341579881.229507649
#Sta/Elev= 30
       0 3257.03      10 3252.39    19.5 3247.31    24.3 3244.15    28.9 3240.82
    33.9 3236.68    50.4 3221.61    57.8 3215.82    62.6 3212.78    66.4 3211.83
    69.3 3211.69    81.7 3211.43    86.5    3212    91.1 3212.08  106.61 3210.28
   114.7 3209.72   124.9 3210.25   133.6    3212   141.8 3212.74   170.9 3213.52
   186.7 3212.98   191.1 3214.43   196.8 3217.61   199.7 3218.24   210.7 3219.01
   222.8 3220.97   234.4 3221.21   241.4 3221.78   248.7  3222.7263.3772 3225.45
#Mann= 4 ,-1,0
       0     .06       0  106.61    .045       0   124.9     .06       0
  184.19      .1       0
#XS Ineff= 2 , 0
                          169.86         3217.56
Permanent Ineff=
       F       F
Bank Sta=106.61,124.9
XS Rating Curve= 0 ,0
Exp/Cntr(USF)=0,0
Exp/Cntr=0.3,0.1

Type RM Length L Ch R = 1 ,8071    ,310.5,304.9,295.7
XS GIS Cut Line= 2
2342837.68545165579567.7422618132342620.79930628579666.265209792
#Sta/Elev= 30
       0 3251.76     5.2 3246.79    19.2 3234.57    32.4 3225.72    54.4 3206.21
    58.8 3202.63    61.5 3201.08    63.2 3200.32    67.6 3199.74    93.9 3200.58
    98.3 3200.28  101.56 3199.36   107.1 3198.62   115.9 3198.72   120.3 3199.39
   124.7  3201.8   129.1 3202.87   146.6 3202.34   155.4 3202.58   164.2 3203.88
     173 3204.21   183.5  3207.1   186.2 3206.92   190.6 3204.98     195 3204.03
   199.4 3204.73   208.1 3205.12   228.8 3204.79   231.8 3205.64 238.215 3209.37
#Mann= 4 ,-1,0
       0      .1       0  101.56    .045       0   120.3      .1       0
     190     .06       0
Bank Sta=101.56,120.3
XS Rating Curve= 0 ,0
Exp/Cntr(USF)=0,0
Exp/Cntr=0.3,0.1

Type RM Length L Ch R = 1 ,7766    ,267.2,273.8,279.6
XS GIS Cut Line= 4
2342641.82657917579349.1038436932342582.81455525579388.275618191
2342520.75018526579475.267481036  2342461.229437579521.561396352
#Sta/Elev= 30
       0 3218.12    16.4 3210.35    29.1 3205.36    44.5 3197.27      50 3194.98
    56.1 3193.88    69.2 3193.33    71.9 3192.76    81.8 3189.11    96.5 3189.51
    99.2  3189.1   101.4 3188.48  105.22 3186.34   111.2 3185.37   116.2 3185.49
   119.3 3186.35     126 3188.79   130.9 3189.53   150.6 3188.77   155.5 3189.54
   170.2 3197.47   175.1 3199.35   178.4 3199.29     188 3196.16   205.1 3197.16
     224 3197.53   229.1 3200.48   239.2 3208.08   244.3 3209.08253.0966 3209.54
#Mann= 5 ,-1,0
       0      .1       0  100.83     .06       0  105.22    .045       0
   119.3     .06       0  247.69      .1       0
Bank Sta=105.22,119.3
XS Rating Curve= 0 ,0
Exp/Cntr(USF)=0,0
Exp/Cntr=0.3,0.1

Type RM Length L Ch R = 1 ,7492    ,217.8,224.6,227.1
XS GIS Cut Line= 2
2342549.23874853579164.4369067752342274.01887836579292.126717151
#Sta/Elev= 30
       0 3207.76     5.6 3204.94    14.4 3201.92    18.8 3199.81      32 3190.45
    49.7 3183.04    52.6 3182.39    67.6 3181.98    76.7 3181.11    98.2 3182.29
   120.2 3181.89   127.9 3182.54   133.5 3181.76  141.97 3176.35   145.9 3175.62
   151.1 3175.52   155.5 3176.32     167 3179.32   173.1 3179.63     182 3178.68
   185.1  3178.9   197.1  3181.3   227.3 3185.52   247.4 3187.13   257.4 3187.27
   261.3 3188.45   270.2 3194.36   287.5 3200.73   292.2 3201.49303.3985 3201.86
#Mann= 3 ,-1,0
       0      .1       0  141.97    .045       0   155.5      .1       0
Bank Sta=141.97,155.5
XS Rating Curve= 0 ,0
Exp/Cntr(USF)=0,0
Exp/Cntr=0.3,0.1

Type RM Length L Ch R = 1 ,7267    ,246.8,248.7,250.3
XS GIS Cut Line= 2
2342477.83939151579007.8473511142342161.29979961579077.373011478
#Sta/Elev= 30
       0  3195.5     9.9 3191.73    18.1 3189.54    36.1 3185.29    49.5 3182.95
      59 3178.15    63.1 3176.83    79.5 3176.59    93.2 3174.88   126.8 3176.48
   140.9  3174.6   149.1 3172.15   157.3 3174.33   165.5 3174.62   169.6 3171.99
   173.6 3168.31   177.8 3167.13   183.8 3166.91   190.6 3167.07  196.13 3168.32
   210.7 3175.66   255.6 3179.64   259.7 3182.11     272 3186.36   280.2 3190.36
   287.9  3190.4   291.3 3191.48   300.7 3197.41   308.9  3200.6324.0851 3208.52
#Mann= 5 ,-1,0
       0      .1       0   173.6    .045       0  196.13      .1       0
     220     .06       0     320      .1       0
Bank Sta=173.6,196.13
XS Rating Curve= 0 ,0
Exp/Cntr(USF)=0,0
Exp/Cntr=0.3,0.1

Type RM Length L Ch R = 1 ,7019    ,295.1,290.6,284.8
XS GIS Cut Line= 3
2342412.83572532578790.2263816832342201.99774714578807.749109091
2342093.46988706578831.489578484
#Sta/Elev= 30
       0 3182.17     4.7 3180.36    20.7 3176.45    47.8 3171.52    56.9  3170.8
    64.9  3168.6    76.9  3166.5     105 3163.94   121.1 3164.34   145.2 3162.64
   153.2 3158.94   157.2    3158   166.4 3158.86   169.2    3160   173.3 3163.28
   177.3 3164.95   181.3  3165.6   201.4  3167.5   225.7 3168.37   233.9 3167.15
   246.2 3160.42   250.3 3159.66   254.4 3159.95   258.5  3161.1   266.7 3164.77
   274.8 3170.55     283 3175.42   295.3 3184.25   299.4  3186.4 322.659 3193.69
#Mann= 5 ,-1,0
       0      .1       0     150     .06       0   153.2    .045       0
   166.4     .06       0  241.56      .1       0
#XS Ineff= 2 , 0
                          209.61         3172.59
Permanent Ineff=
       F       F
Bank Sta=153.2,166.4
XS Rating Curve= 0 ,0
Exp/Cntr(USF)=0,0
Exp/Cntr=0.3,0.1

Type RM Length L Ch R = 1 ,6728    ,241.9,246.7,250.4
XS GIS Cut Line= 3
2342433.18469908578497.9925084462342256.26167718578560.169928283
2342071.42516548578568.083418081
#Sta/Elev= 30
       0 3211.99    13.8 3207.02    34.7 3196.15    68.9 3182.43    78.6 3177.43
      82 3175.35      88 3170.14    98.6 3159.89   107.6 3149.94   111.3 3148.43
   115.5 3148.32     124 3148.46   127.2 3149.71   132.5 3151.03     157 3151.39
   162.2 3153.74   166.4 3154.84   183.4 3155.27   199.6  3154.2   219.6 3157.14
   230.8 3157.81   251.7 3158.02   259.7 3157.04   267.7 3158.86   283.7 3157.85
   319.1 3159.58   334.5 3161.94   343.8 3162.55   363.8 3167.21372.5366 3170.22
#Mann= 5 ,-1,0
       0      .1       0   107.6    .045       0   127.2      .1       0
     180     .06       0  372.54      .1       0
Bank Sta=107.6,127.2
XS Rating Curve= 0 ,0
Exp/Cntr(USF)=0,0
Exp/Cntr=0.3,0.1

Type RM Length L Ch R = 1 ,6481    ,354.2,356.6,354.6
XS GIS Cut Line= 4
2342383.00495687578339.3803644722342342.17112983578310.299678693
2342263.60991771578305.2425069492342060.68542933 578305.80775622
#Sta/Elev= 30
       0 3189.07    23.1 3180.29    35.2 3174.48    45.2 3168.12    72.2 3147.97
    80.2 3144.12    84.2 3143.38   100.2 3144.12   108.2 3142.23   112.3 3141.93
   120.3  3143.5   128.2 3143.69   136.4 3143.24     1423142.162   148.3 3141.22
   152.4 3141.23   157.33142.227   164.3 3145.13   172.3  3146.6   180.5 3147.36
     204 3147.52   216.3 3146.36   224.3 3147.92   228.3 3148.06   260.3 3146.89
   276.8 3147.51   292.3  3149.8   304.3 3152.22   316.3 3155.47   331.8 3158.24
#Mann= 5 ,-1,0
       0      .1       0     110     .06       0     142    .045       0
   157.3     .06       0  201.56      .1       0
Bank Sta=142,157.3
XS Rating Curve= 0 ,0
Exp/Cntr(USF)=0,0
Exp/Cntr=0.3,0.1

Type RM Length L Ch R = 1 ,6125    ,240.5,245.4,250.3
XS GIS Cut Line= 3
2342486.31813058578002.2688975592342339.91856933577979.093677438
 2342016.0307369577979.093677438
#Sta/Elev= 30
       0 3175.79    18.4 3167.14    34.6 3160.64    58.9 3148.47    83.2 3141.13
   115.6 3138.46   148.2 3138.34     172 3136.44     184 3133.85     196 3128.83
     200 3127.54     204 3127.41     212 3127.58     216 3128.95     232 3135.02
     244 3136.28     292 3137.08     308 3136.65     316 3135.66     324 3133.36
     332 3132.85     336 3133.79     348 3139.26     364 3143.33     392 3152.23
     408 3158.38     428 3163.99     440  3169.2     448  3171.3472.1104 3182.32
#Mann= 5 ,-1,0
       0      .1       0      20     .06       0     196    .045       0
     216     .06       0  318.22      .1       0
Bank Sta=196,216
XS Rating Curve= 0 ,0
Exp/Cntr(USF)=0,0
Exp/Cntr=0.3,0.1

Type RM Length L Ch R = 1 ,5879    ,273.2,276.2,278.4
XS GIS Cut Line= 3
2342529.94872332577842.080820817  2342276.214606577732.799295042
2342047.60267852577727.146802329
#Sta/Elev= 30
       0 3159.73    10.6 3153.98    41.6  3141.3    54.2  3134.7    71.6 3131.28
    93.4 3124.96   115.2 3123.39   128.2 3124.55   163.1 3124.94   197.9 3123.43
     211 3123.92   233.4 3122.89   251.7 3120.95   263.2 3120.33   265.2 3120.97
     272 3124.71   288.3 3124.25   304.3  3122.3   312.3  3122.6   320.3 3124.62
   328.3 3124.98   340.3 3130.45   348.3 3131.64   384.3 3130.26   392.3 3133.08
   400.3 3134.39   420.4 3139.84   448.4 3148.96   476.4 3158.83504.9488  3170.7
#Mann= 6 ,-1,0
       0     .06       0     180      .1       0   251.7    .045       0
   265.2      .1       0  286.27     .06       0  386.27      .1       0
#XS Ineff= 2 , 0
          164.28  3129.2  277.08         3132.73
Permanent Ineff=
       F       F
Bank Sta=251.7,265.2
XS Rating Curve= 0 ,0
Exp/Cntr(USF)=0,0
Exp/Cntr=0.3,0.1

Type RM Length L Ch R = 1 ,5603    ,275.6,264,251.2
BEGIN DESCRIPTION:
The IFA is very tricky here
END DESCRIPTION:
XS GIS Cut Line= 3
2342581.44921248577619.1213860462342372.30698211577463.991863825
2342092.82262022 577475.29684925
#Sta/Elev= 30
       0 3135.01    46.4 3122.05    71.3 3119.83    81.3 3117.61    97.3 3117.89
   119.5 3115.06     151 3112.84   184.5 3113.12   195.8 3111.55   208.9 3111.52
   215.7 3112.36   248.2 3112.38   260.5 3114.39   272.5    3113   284.5 3113.33
   296.6 3109.27   336.6 3112.77   360.6 3111.51   368.6 3107.62   372.6 3107.09
   384.8 3109.04   392.6 3111.58   412.7 3113.02   428.7 3123.41   436.7 3126.28
   460.7  3126.7   488.8 3124.46   496.4    3128   512.7  3137.7540.1081 3144.74
#Mann= 6 ,-1,0
       0     .06       0    81.3      .1       0   195.8    .045       0
   208.9      .1       0   360.6     .06       0   460.7      .1       0
#XS Ineff= 2 , 0
                          260.13         3119.79
Permanent Ineff=
       F       F
Bank Sta=195.8,208.9
XS Rating Curve= 0 ,0
Exp/Cntr(USF)=0,0
Exp/Cntr=0.3,0.1

Type RM Length L Ch R = 1 ,5339    ,354.6,350.9,340.7
XS GIS Cut Line= 3
2342713.96876385577222.1907866792342434.85686193577288.446463824
2342098.23188718577339.198887471
#Sta/Elev= 30
       0 3137.46    47.1 3127.59    55.3 3124.23    73.7 3112.94    88.2  3106.8
   121.1 3107.15   134.2 3102.84   166.3 3105.27   207.4 3103.95   220.23101.814
   232.1 3101.21   240.83101.652   256.7 3102.12   273.2 3106.32   281.4 3107.25
   321.9 3106.03   370.5 3107.24   398.8 3104.47   409.4 3102.05   425.9 3101.36
   463.5 3105.26   471.6 3104.37   493.8 3105.57   524.2 3105.18   536.9 3109.51
   552.5 3118.53   560.5 3121.55   584.9 3122.15   613.2    3120   627.3 3129.18
#Mann= 5 ,-1,0
       0      .1       0   220.2    .045       0   240.8      .1       0
  567.81     .06       0  577.81      .1       0
#XS Ineff= 2 , 0
          163.27 3110.85  362.79         3109.73
Permanent Ineff=
       F       F
Bank Sta=220.2,240.8
XS Rating Curve= 0 ,0
Exp/Cntr(USF)=0,0
Exp/Cntr=0.3,0.1

Type RM Length L Ch R = 1 ,4988    ,165.1,165.2,163.3
XS GIS Cut Line= 4
2342493.62234599576852.645754917 2342342.0918063576994.270896907
2342313.95636471 577013.712893942342087.78209199577188.387571372
#Sta/Elev= 30
       0 3119.55    35.9 3110.14    69.3 3098.17   102.9 3092.81   117.4 3091.65
   129.7 3093.21   145.7 3091.35   160.8 3093.84   171.2    3094   188.1 3092.53
   214.6 3092.85   224.3 3091.38   240.7 3092.31   248.9  3091.4   262.5 3090.66
   269.1 3091.33   299.5 3093.74   332.4 3091.47   370.2 3094.48   390.8    3095
     405 3093.82   410.7  3095.2   425.8 3095.24   436.4 3096.98   451.1 3096.81
   456.4    3098   466.2 3102.98   481.4 3107.33   493.4 3114.58   527.4 3116.43
#Mann= 4 ,-1,0
       0      .1       0   248.9    .045       0   269.1      .1       0
     448     .06       0
#XS Ineff= 2 , 0
          130.56 3097.39  304.98         3096.87
Permanent Ineff=
       F       F
Bank Sta=248.9,269.1
XS Rating Curve= 0 ,0
Exp/Cntr(USF)=0,0
Exp/Cntr=0.3,0.1

Type RM Length L Ch R = 1 ,4823    ,171.8,170,166.9
XS GIS Cut Line= 3
2342380.12363185576770.4264379812342108.46773509576984.491284624
2342006.32511791577076.854289521
#Sta/Elev= 30
       0 3117.05    21.9 3107.76    50.3 3097.78    87.4 3088.61   101.8 3088.28
   115.9  3086.5   142.5  3088.3   152.9 3088.64   162.9 3087.79   178.2 3088.54
   203.6 3085.59   232.6 3088.39   264.8 3087.32   272.5 3085.74     280 3085.11
   284.5 3085.73   292.4 3088.04   300.4 3086.52   308.2 3086.14   320.9 3088.29
   346.3 3088.14   362.4 3089.76   377.7 3089.72   389.4 3094.13   400.4  3094.8
   405.6 3096.07   420.2 3105.85   427.1 3108.18   459.5 3109.79   483.6 3108.37
#Mann= 4 ,-1,0
       0      .1       0   272.5    .045       0   284.5      .1       0
   427.1     .06       0
#XS Ineff= 2 , 0
          137.87 3092.94  329.73          3094.3
Permanent Ineff=
       F       F
Bank Sta=272.5,284.5
XS Rating Curve= 0 ,0
Exp/Cntr(USF)=0,0
Exp/Cntr=0.3,0.1

Type RM Length L Ch R = 1 ,4653    ,89.1,89.8,87.7
XS GIS Cut Line= 2
2342250.81542499576616.1258886242341919.39523095576968.191930819
#Sta/Elev= 30
       0 3118.06    34.4 3103.54    56.4 3090.47    70.5 3086.01    97.2 3080.92
   108.9 3082.36   144.3 3081.62   166.3 3078.57   178.1 3081.92   190.6    3081
   231.4 3083.08   254.8 3081.07   274.3 3080.92     284 3081.85   298.1 3080.69
   319.5 3082.25   330.23081.399  345.48 3081.31   359.8 3083.44   391.5 3082.33
   407.3 3084.98   413.5 3087.03   429.9 3098.16   429.9 3098.18   429.9  3098.2
   435.4  3099.7   446.4 3100.59   476.5 3098.72   479.4 3099.33   483.5  3101.9
#Mann= 4 ,-1,0
       0      .1       0   330.2    .045       0  345.48      .1       0
   429.9     .06       0
#XS Ineff= 2 , 0
           149.5 3087.94   362.7         3086.01
Permanent Ineff=
       F       F
Bank Sta=330.2,345.48
XS Rating Curve= 0 ,0
Exp/Cntr(USF)=0,0
Exp/Cntr=0.3,0.1

Type RM Length L Ch R = 1 ,4563    ,196.3,200.4,197.7
XS GIS Cut Line= 3
2342186.01928685576551.588661202 2341984.4214672576807.462816913
 2341860.3612705576947.805914439
#Sta/Elev= 30
       0 3116.61    28.1 3103.98    39.5 3100.57    52.9 3094.56    61.2 3092.83
    76.5  3083.5    98.8 3078.44   106.4 3078.34   119.2 3080.13   129.3 3078.29
   159.1 3079.53   190.4 3077.31   216.1 3080.67   235.7 3076.47   270.2 3081.13
   274.4 3080.58  279.85  3077.9   284.4 3077.08   293.8 3077.88   319.7 3080.33
   349.8 3081.26   406.5 3080.45   413.5 3083.62   428.8  3094.4   434.8 3095.91
   456.2 3095.71   477.1 3093.79   482.9 3094.95   497.2 3105.65513.0659 3113.58
#Mann= 5 ,-1,0
       0      .1       0  279.85    .045       0   293.8      .1       0
  345.75     .06       0  485.75      .1       0
#XS Ineff= 2 , 0
          212.29 3085.98  324.51         3083.44
Permanent Ineff=
       F       F
Bank Sta=279.85,293.8
XS Rating Curve= 0 ,0
Exp/Cntr(USF)=0,0
Exp/Cntr=0.3,0.1

Type RM Length L Ch R = 1 ,4363    ,204.2,204.1,196.9
XS GIS Cut Line= 2
2342020.86414999576448.4636226892341731.64881641576840.028618549
#Sta/Elev= 30
       0 3112.74    35.7 3097.11    58.2 3083.68    75.4 3075.36    80.5 3073.84
    95.4 3073.59   106.8 3075.54   115.3 3075.11   122.3  3073.4   142.5 3074.48
     170 3072.94   192.6  3076.8   244.6 3074.77   249.5 3074.17   254.5 3071.88
   261.3 3071.28   272.7 3069.95   279.4 3071.19   324.1  3074.5   367.1 3074.57
   372.8 3076.19   387.1 3085.07   395.7 3085.82     410 3084.76   427.2 3082.79
   438.6 3078.26   452.9 3078.29     459 3080.42   475.7 3092.54486.7943 3096.55
#Mann= 5 ,-1,0
       0      .1       0   261.3    .045       0   279.4      .1       0
     410     .06       0     420      .1       0
#XS Ineff= 2 , 0
           196.9  3080.5
Permanent Ineff=
       F       F
Bank Sta=261.3,279.4
XS Rating Curve= 0 ,0
Exp/Cntr(USF)=0,0
Exp/Cntr=0.3,0.1

Type RM Length L Ch R = 1 ,4159    ,392.1,392.3,382.9
XS GIS Cut Line= 3
2341896.97913679576360.2713995272341729.49787123576567.296852784
2341596.13315977576785.952949482
#Sta/Elev= 30
       0 3109.87    21.1 3101.59    37.2 3096.84    58.5 3085.43    77.6 3070.93
      84 3068.37    96.7 3068.98   137.7    3066   160.5 3070.32   192.1 3068.95
   211.7 3070.49   251.5 3070.01   268.5  3071.1   277.9 3070.66     289 3068.27
   301.3 3068.44   312.3 3065.79   338.8 3065.67   344.3 3065.11     353 3065.66
   358.8 3068.92   366.9 3070.68   376.3 3075.66   382.1 3076.58   408.3 3075.55
   437.2 3071.82   454.9 3073.09   475.2    3083   512.1 3089.66522.4068 3092.51
#Mann= 5 ,-1,0
       0      .1       0   338.8    .045       0     353      .1       0
  366.29     .06       0  522.41      .1       0
#XS Ineff= 2 , 0
          212.62 3074.64
Permanent Ineff=
       F       F
Bank Sta=338.8,353
XS Rating Curve= 0 ,0
Exp/Cntr(USF)=0,0
Exp/Cntr=0.3,0.1

Type RM Length L Ch R = 1 ,3767    ,290.6,291.1,289.6
XS GIS Cut Line= 3
 2341644.6671179 576122.06116933 2341439.8146326576336.486200677
2341322.07231628576626.534345759
#Sta/Elev= 30
       0 3096.02    16.7 3091.44    70.7 3085.49   115.7 3078.91   128.1 3076.22
   137.1 3071.74   145.5 3069.11   162.8 3069.15     186 3063.07   228.9 3060.48
     243 3057.91   267.1 3057.28   297.3 3059.04   356.6 3054.95     375 3054.94
  383.16  3052.1   391.3 3051.39   407.5 3052.08   418.2 3051.93   431.1  3055.2
   447.3 3054.71     457 3058.11   468.8 3059.96   487.4  3060.8   534.7 3055.66
   569.3 3057.25   577.9 3060.56   585.4 3065.39   590.9 3067.58609.5867 3071.47
#Mann= 7 ,-1,0
       0      .1       0   356.6     .06       0  383.16    .045       0
   407.5     .06       0   447.3      .1       0   468.8     .06       0
   577.9      .1       0
Bank Sta=383.16,407.5
XS Rating Curve= 0 ,0
Exp/Cntr(USF)=0,0
Exp/Cntr=0.3,0.1

Type RM Length L Ch R = 1 ,3476    ,213.6,210.1,201.3
XS GIS Cut Line= 3
2341213.44405553576193.3888555132341125.42754498576384.091295035
2341099.02259181576576.749657014
#Sta/Elev= 30
       0 3058.85    24.9 3057.73      43 3054.22    52.6 3056.61    61.1 3056.68
    83.5  3051.4   105.5  3050.1  113.75 3046.19   127.1 3045.65   133.4 3046.21
   140.7 3048.07   149.6 3049.04   167.2 3049.23   180.4 3047.95   193.6 3050.19
   212.1  3049.7   231.3 3051.01   247.6 3050.76   267.7 3053.38   300.9 3050.64
     304 3050.21   312.1 3047.17   320.1  3046.6   324.2 3046.92   336.3 3051.22
   350.6 3050.89   376.7 3052.84   380.7 3054.07   388.8 3058.02   404.5 3068.07
#Mann= 4 ,-1,0
       0      .1       0  113.75    .045       0   133.4      .1       0
   300.9     .06       0
#XS Ineff= 2 , 0
                          194.35         3057.22
Permanent Ineff=
       F       F
Bank Sta=113.75,133.4
XS Rating Curve= 0 ,0
Exp/Cntr(USF)=0,0
Exp/Cntr=0.3,0.1

Type RM Length L Ch R = 1 ,3266    ,194.2,197.5,196.5
XS GIS Cut Line= 3
2341023.71957723576134.7111818142340964.06394231 576258.91225781
2340959.17413617 576497.53479752
#Sta/Elev= 30
       0 3072.05    25.5 3067.97    35.9 3066.97    45.1 3065.02      56 3063.62
      66  3061.7   100.4 3056.44   104.8 3055.63   113.7 3053.06   118.1 3052.44
   127.4 3052.52   135.9 3051.87   160.1 3048.38   164.1 3048.16   168.1 3047.42
   176.1 3042.77   180.1 3041.78   192.1 3041.45   214.4 3041.79   228.1 3044.47
   244.1 3044.49   256.1 3045.76   280.1 3045.96   288.1 3046.98   296.1 3049.19
   308.1 3049.11   340.4 3046.76   348.1 3045.83   360.1 3047.55   376.5 3047.74
#Mann= 3 ,0,0
       0      .1       0   180.1    .045       0   214.4      .1       0
Bank Sta=180.1,214.4
XS Rating Curve= 0 ,0
Exp/Cntr(USF)=0,0
Exp/Cntr=0.3,0.1

Type RM Length L Ch R = 1 ,3068    ,307.5,311.8,310.4
XS GIS Cut Line= 3
2340795.58228395 576083.770985162340771.65091885576210.128592919
2340778.35170108576524.108103106
#Sta/Elev= 30
       0 3062.52    13.6 3060.66    38.1 3055.78    62.3 3053.07    99.1  3046.8
   123.6 3043.61   135.7 3043.94   147.7 3042.23   163.7 3042.04   175.7 3039.09
   187.7 3039.07   196.6 3036.49   203.7  3035.5   211.7  3035.6     217 3036.56
   239.7 3041.41   259.7 3040.99   274.3 3038.75   295.7 3037.81   307.7 3039.94
   327.7 3039.98   331.7 3040.46   339.7 3043.19   351.7 3044.16   391.7  3041.7
   399.7 3043.46   407.7  3043.5   418.1 3045.22   427.7  3048.4442.6549 3051.83
#Mann= 4 ,-1,0
       0      .1       0   196.6    .045       0     217      .1       0
   408.6     .06       0
#XS Ineff= 2 , 0
                          250.83         3044.88
Permanent Ineff=
       F       F
Bank Sta=196.6,217
XS Rating Curve= 0 ,0
Exp/Cntr(USF)=0,0
Exp/Cntr=0.3,0.1

Type RM Length L Ch R = 1 ,2756    ,354.4,346.1,338.6
XS GIS Cut Line= 3
2340495.96159283576093.3435312032340481.60277376576430.297151892
2340529.46550398576584.415143172
#Sta/Elev= 30
       0 3055.68    19.9 3052.93    43.9 3046.18    55.9 3043.95    87.9 3040.09
   115.9 3035.72     160 3034.63     172 3032.49     180 3033.44     188 3032.65
     208 3033.18     224 3032.77     236 3031.45   240.1 3029.22   242.6 3028.55
   248.1 3027.83  261.93 3028.56   272.1 3031.32   280.1 3030.34   304.1 3029.83
   316.1 3032.63   324.1 3033.53   340.3 3033.42   369.6 3035.26   386.4 3034.66
   403.1 3036.51   436.6 3036.13   447.1 3039.72   469.5 3044.08498.6385 3051.74
#Mann= 4 ,-1,0
       0      .1       0   242.6    .045       0  261.93      .1       0
  407.26     .06       0
#XS Ineff= 2 , 0
                          299.83         3037.04
Permanent Ineff=
       F       F
Bank Sta=242.6,261.93
XS Rating Curve= 0 ,0
Exp/Cntr(USF)=0,0
Exp/Cntr=0.3,0.1

Type RM Length L Ch R = 1 ,2410    ,270.9,275.4,278.7
XS GIS Cut Line= 2
2340063.28251172576228.3164303992340276.75028846576640.893164822
#Sta/Elev= 30
       0 3067.65    32.5 3052.95      46 3048.21    69.6 3035.84      82 3027.76
    87.4 3026.14    97.7 3024.42   113.6 3023.47     126 3025.03   145.1 3024.36
   158.6 3022.13     176 3023.72   191.3 3023.27   226.2 3024.04   238.7 3022.18
   257.7 3021.59   265.5 3022.23   271.8 3025.46   284.7 3027.14   316.2 3026.48
   332.7 3025.14   372.3 3026.15   379.3 3024.86   390.1 3027.63   401.8 3028.96
   424.3 3029.42   434.6 3028.88   440.6 3030.26   451.3 3035.58464.5299 3038.24
#Mann= 6 ,-1,0
       0      .1       0     190     .07       0   238.7    .045       0
   265.5     .07       0     300     .06       0     410      .1       0
#XS Ineff= 2 , 0
          128.78 3026.96
Permanent Ineff=
       F       F
Bank Sta=238.7,265.5
XS Rating Curve= 0 ,0
Exp/Cntr(USF)=0,0
Exp/Cntr=0.3,0.1

Type RM Length L Ch R = 1 ,2134    ,95.1,95.2,94
XS GIS Cut Line= 3
2339926.73008521576240.3531045472339904.67962373576440.040823478
2340011.06727361576751.612264651
#Sta/Elev= 30
       0 3088.37    45.1 3064.95    73.3 3046.08    77.3 3042.85    93.4 3027.17
    97.4 3023.91   104.5 3020.61   121.6 3019.26   177.9 3020.71   185.9 3019.61
   223.2 3019.22   227.5 3018.87   231.13017.218   235.9 3016.62   248.5 3017.18
     277 3018.41   324.3 3016.47   349.5 3017.93   362.7 3016.09   375.4 3016.47
   392.3 3014.57   413.4  3016.8   430.3 3017.61     444 3021.35   455.7 3022.68
   472.4 3022.92   485.3 3021.97     498 3025.67   519.1 3026.54   530.1 3029.53
#Mann= 6 ,-1,0
       0      .1       0   211.4     .07       0   231.1    .045       0
   248.5     .07       0   338.5     .06       0   452.5      .1       0
#XS Ineff= 2 , 0
          173.42 3025.34  373.52          3029.8
Permanent Ineff=
       F       F
Bank Sta=231.1,248.5
XS Rating Curve= 0 ,0
Exp/Cntr(USF)=0,0
Exp/Cntr=0.3,0.1

Type RM Length L Ch R = 1 ,2039    ,115.8,116.1,115.9
XS GIS Cut Line= 3
2339913.90746094576190.6959305212339794.41477372576399.479856546
2339936.23027065576788.159366631
#Sta/Elev= 30
       0  3106.6    16.7 3102.83    44.1 3094.18    59.9 3090.36    85.8 3078.58
   118.1 3061.69   164.5 3027.71   173.4 3022.01   182.6  3018.3   196.4 3016.84
   233.3 3019.74   276.4 3016.76   289.2 3017.56   357.3 3017.16   365.8 3015.61
   377.4 3015.52   387.1 3017.28   425.5 3014.85   459.5 3017.06   472.3 3015.42
   490.8 3017.19   505.3 3016.54   519.1  3012.8   530.3 3013.95   542.7 3013.66
   561.7 3019.12   570.2 3020.15   592.7 3020.73   608.6 3019.01654.3034 3029.64
#Mann= 6 ,-1,0
       0      .1       0   365.8    .045       0   377.4      .1       0
  450.56     .08       0  550.56     .06       0  650.56      .1       0
#XS Ineff= 2 , 0
           235.1 3021.79  513.86         3022.01
Permanent Ineff=
       F       F
Bank Sta=365.8,377.4
XS Rating Curve= 0 ,0
Exp/Cntr(USF)=0,0
Exp/Cntr=0.3,0.1

Type RM Length L Ch R = 1 ,1923    ,196.5,196.3,195.1
XS GIS Cut Line= 3
2339816.45469621576229.2462347822339688.94838293576440.320875015
2339836.26986652576861.608626338
#Sta/Elev= 30
       0 3056.85    23.3 3048.62    64.2 3036.27   126.1  3018.5   140.1 3015.66
   246.7 3014.37   272.9 3012.22   285.6 3013.63   311.1 3013.19   365.4 3014.56
  372.97 3013.85   384.8 3013.83   391.6 3014.74   412.8 3013.63   425.6 3014.22
   450.9 3013.23   510.4 3015.16   516.7 3014.31   526.1 3010.69   548.4 3009.66
   554.3 3010.31   565.3 3015.76     570 3016.88     592 3017.84   607.7 3016.53
   620.7 3018.26   628.9 3018.42   644.1 3021.49   656.3 3022.54   692.9 3029.69
#Mann= 6 ,-1,0
       0      .1       0  372.97    .045       0   384.8      .1       0
   425.6     .08       0   526.1     .06       0   620.7      .1       0
#XS Ineff= 2 , 0
           231.4 3021.66  512.45         3017.02
Permanent Ineff=
       F       F
Bank Sta=372.97,384.8
XS Rating Curve= 0 ,0
Exp/Cntr(USF)=0,0
Exp/Cntr=0.3,0.1

Type RM Length L Ch R = 1 ,1727    ,137,138.7,137.7
XS GIS Cut Line= 4
2339753.70847368576260.2905725292339628.96336065576385.035685563
 2339543.6114412576551.8002050932339694.61868329576931.287970007
#Sta/Elev= 30
       0 3032.55    19.1 3030.73    52.6 3024.89    64.4 3023.82   200.9  3018.4
     262 3014.26   279.9 3014.09   306.9 3010.42   319.8  3009.7   347.3 3010.81
   360.8 3009.33   386.8 3008.97   395.4 3008.02  407.72 3008.02   416.9 3009.44
   451.8 3008.12   482.3 3009.31   519.2 3007.58   528.5 3008.05   537.4 3006.92
   550.4 3009.27     559 3009.74   584.8    3009   593.4 3006.05   597.7 3005.75
   610.6  3010.7   632.2 3013.32   731.7 3014.36   747.1 3016.94772.1827 3019.48
#Mann= 6 ,-1,0
       0      .1       0  296.42     .08       0   395.4    .045       0
  407.72     .08       0  563.75     .06       0  723.75      .1       0
#XS Ineff= 2 , 0
          343.44  3012.5  580.12         3012.67
Permanent Ineff=
       F       F
Bank Sta=395.4,407.72
XS Rating Curve= 0 ,0
Exp/Cntr(USF)=0,0
Exp/Cntr=0.3,0.1

Type RM Length L Ch R = 1 ,1588    ,124.6,122.2,121.8
XS GIS Cut Line= 5
2339259.28112726576579.1603487872339389.79165014576626.515236985
2339431.70818718 576629.650888232339515.70890161576852.025767329
2339659.50203567577030.681466664
#Sta/Elev= 30
       0 3066.81     9.5 3066.28      18 3063.15      52 3041.56    64.8 3035.31
    90.3 3013.66   102.2  3007.3   115.8 3004.12   127.2 3004.92   141.2 3007.37
   145.2 3007.29   153.3  3004.8   157.3 3004.58   180.9 3006.47   193.2 3004.46
   202.6 3004.02   210.3    3004   257.3  3002.4   270.2 3003.44     283  3001.4
     305 3004.15   326.7 3004.33   347.1 3007.09   398.1 3007.74   415.5 3010.53
   440.6 3010.83   461.1 3009.02   527.9 3010.04   621.7 3018.68   647.9 3024.56
#Mann= 8 ,-1,0
       0     .06       0   134.1      .1       0   202.6    .045       0
   210.3      .1       0   401.3     .08       0     452     .06       0
   509.6     .07       0   573.3      .1       0
#XS Ineff= 2 , 0
          140.79 3013.37  347.86          3012.8
Permanent Ineff=
       F       F
Bank Sta=202.6,210.3
XS Rating Curve= 0 ,0
Exp/Cntr(USF)=0,0
Exp/Cntr=0.3,0.1

Type RM Length L Ch R = 1 ,1466    ,245.9,239.2,229.9
XS GIS Cut Line= 5
2339257.17565197576655.2191562242339370.13169527 576697.33835881
2339483.08773857576877.3022244052339568.28339835577011.317868998
2339625.70697312577080.339267739
#Sta/Elev= 30
       0  3056.1    20.3 3042.95    28.8 3035.23    37.4 3028.99      63 3006.23
      66 3004.45    72.3 3003.02    90.3 3003.03    97.1 3002.72   105.7 3005.07
   109.9 3005.18   139.3 3003.37     162 3003.41   175.9 3001.67   181.8 3000.57
   194.5 3001.57   200.6 3003.23   220.6  3002.8   232.2 3001.33   247.9 3002.26
   264.1 3005.55   313.4 3009.37   347.1 3009.29   356.9 3007.88     404 3007.77
   441.9 3008.34   464.1 3010.45   490.2 3011.38   530.7 3016.07   581.6 3025.19
#Mann= 8 ,-1,0
       0     .06       0    90.3      .1       0   175.9    .045       0
   194.5      .1       0   220.6     .08       0   347.1     .06       0
     404     .07       0   464.1      .1       0
#XS Ineff= 2 , 0
          107.83 3011.08
Permanent Ineff=
       F       F
Bank Sta=175.9,194.5
XS Rating Curve= 0 ,0
Exp/Cntr(USF)=0,0
Exp/Cntr=0.3,0.1

Type RM Length L Ch R = 1 ,1227    ,198.3,167,101.5
BEGIN DESCRIPTION:
xs 4
END DESCRIPTION:
XS GIS Cut Line= 4
2339118.37373436576767.2179449192339272.49172564 576896.44731649
2339430.43873534576836.1402764232339619.01789237577093.641764961
#Sta/Elev= 30
       0 3059.68    19.7 3056.64    31.1 3051.11    42.4 3050.67    48.1 3049.27
    73.7  3029.2    87.9 3013.14    99.2 3002.74   104.9 2998.67   110.6 2996.59
   136.1 2995.79   144.6 2996.59   167.4 2999.42   183.6 2998.06     196 3000.02
   243.4 3000.83     265 3002.73   282.1 3001.38   373.1 3003.28   406.5 3008.51
   422.5 3009.52   440.9 3009.06   455.2 3005.58   467.9 3007.22   489.5 3007.86
   500.4 3006.81   520.2 3007.04   610.1 3012.79   644.1 3017.22689.3663 3025.15
#Mann= 10 ,-1,0
       0      .1       0      10     .06       0   110.6    .045       0
   144.6      .1       0     190     .06       0  241.13      .1       0
  261.13     .08       0   430.2     .06       0   520.2     .07       0
   560.2      .1       0
Bank Sta=110.6,144.6
XS Rating Curve= 0 ,0
Exp/Cntr(USF)=0,0
Exp/Cntr=0.5,0.3

Type RM Length L Ch R = 1 ,1060    ,146.3,171.3,224.6
BEGIN DESCRIPTION:
xs 3
END DESCRIPTION:
XS GIS Cut Line= 6
2338774.71933144577065.8813814382338821.62480705577078.325691293
2338902.99144841577063.0096176262339179.63802903 576939.52377368
2339414.16540707576861.9861507382339595.08652727577110.872347837
#Sta/Elev= 30
       0 3007.87     7.2 3007.66    13.9 3005.13    48.5 2997.52   249.5 3002.54
   285.1 3000.53   327.2 2994.99   345.2 2993.34   411.8 2995.11   452.6 2999.26
   472.1 2997.49   502.6 3000.08     561 3000.73   604.6  3002.9   620.7 3001.61
   675.6 3002.59   686.4 3003.64   701.4  3008.1   716.2 3008.96   731.1 3008.76
   745.9 3005.66   765.7 3005.34   781.3 3003.58   794.9 3005.54     825 3007.28
   875.3 3009.71   892.5 3009.08   906.8 3011.69   958.2 3017.47990.3244  3024.4
#Mann= 6 ,-1,0
       0     .06       0   327.2    .045       0   411.8     .06       0
  628.05     .08       0  712.63     .06       0  862.63      .1       0
#XS Ineff= 3 ,-1
   15.77  234.93 3002.97  234.93   292.2 2995.59   446.8990.3244 3002.54
Permanent Ineff=
       F       F       F
Bank Sta=327.2,411.8
XS Rating Curve= 0 ,0
Exp/Cntr(USF)=0,0
Exp/Cntr=0.5,0.3

Type RM Length L Ch R = 1 ,888     ,300,307.1,314.5
BEGIN DESCRIPTION:
xs 2
END DESCRIPTION:
XS GIS Cut Line= 6
2338711.73197848577067.7958906472338798.67509988577130.543992421
2339002.54592725577111.8296024422339041.16851769577125.314268471
2339435.22500836576918.4641723872339582.64221741577117.573130067
#Sta/Elev= 30
       0 3001.97      16 3001.83    36.5 2994.34    43.4 2993.86    84.4 2996.69
    98.1  2995.6   112.7 2999.84   156.8 3006.68   225.2 3008.58   233.3 3006.69
   245.4 3000.92   297.9 2996.51     3162992.126   327.1 2990.89   347.52992.087
   373.4 2994.62   397.7 3000.31   414.1 2999.23   505.9 3001.08   543.4    3006
   577.1 2999.92   601.5  2998.8   660.4 2999.77   685.5 3001.96   797.9 3005.56
   853.3  3003.5   887.2 3006.69   953.4 3009.52  1013.5 3015.82    1047 3022.44
#Mann= 8 ,-1,0
       0     .06       0  137.22      .1       0     316    .045       0
   347.5      .1       0  452.05     .07       0  559.88      .1       0
  651.33     .06       0  939.22      .1       0
#XS Ineff= 3 ,-1
   10.82  136.56 3002.27  136.56     290    2994   373.5    1047    3002
Permanent Ineff=
       F       F       F
Bank Sta=316,347.5
XS Rating Curve= 0 ,0
Exp/Cntr(USF)=0,0
Exp/Cntr=0.5,0.3

Type RM Length L Ch R = 1 ,581     ,234.6,241.7,240.9
XS GIS Cut Line= 6
2338664.57330325577052.7584464512338640.04582477577158.164792367
 2338789.0781505577298.494250266 2338915.2079854577398.881743966
2339051.42803193577396.8158314532339274.74874767577345.966597476
#Sta/Elev= 30
       0 2993.89    16.9 2996.41    29.2 2994.53    41.5 2990.46    78.5 2992.81
    90.8 2990.84   112.6 2990.35   124.6 2988.72   229.3 2989.22   256.7 2990.43
   291.5 2986.89   306.2 2990.15   349.4 2991.12   362.9  2990.8   377.22987.286
   387.9 2986.35  397.67 2987.23   407.2 2990.33   432.9  2991.8   483.1 2991.67
   499.1 2989.54   527.1 2988.65   547.1 2991.95     591 2993.96   674.2 2994.51
   721.9  2996.7   770.9 2996.59   795.7 3000.38   828.6 3001.17   839.4  3003.6
#Mann= 6 ,-1,0
       0     .06       0     150      .1       0   377.2    .045       0
  397.67      .1       0  599.09     .06       0  765.67      .1       0
#XS Ineff= 2 , 0
           141.2 2994.87  456.34         2993.73
Permanent Ineff=
       F       F
Bank Sta=377.2,397.67
XS Rating Curve= 0 ,0
Exp/Cntr(USF)=0,0
Exp/Cntr=0.3,0.1

Type RM Length L Ch R = 1 ,340     ,281.9,281.9,281.9
XS GIS Cut Line= 6
 2338626.2361811577033.8354169162338604.82854581577130.325002913
2338643.57545066577414.3220573782338850.34244517577667.994527499
2339027.43454696577597.1576867862339159.53568234577600.029450599
#Sta/Elev= 30
       0 2996.76    36.2 2994.11    60.8 2989.09    97.7 2991.86   121.9 2987.99
   247.1  2987.8   271.3  2986.5   283.4 2984.51   335.9 2986.19     352 2984.29
   364.1 2987.46   399.1 2987.36     415 2985.38   437.1  2986.5     551 2985.81
   569.8 2983.01   581.2  2981.9   589.8 2983.08   605.9 2985.62   675.1 2985.13
   746.9 2987.14   760.3 2982.91   765.2 2982.63     776 2987.67   834.2 2988.83
   904.5 2992.39   941.3 2993.36   985.3 2997.29  1003.1 3003.18  1036.6 3009.71
#Mann= 6 ,-1,0
       0     .06       0  148.84      .1       0   569.8    .045       0
   589.8      .1       0  685.46     .06       0   904.5      .1       0
#XS Ineff= 2 , 0
          366.78 2992.88  655.81         2993.39
Permanent Ineff=
       F       F
Bank Sta=569.8,589.8
XS Rating Curve= 0 ,0
Exp/Cntr(USF)=0,0
Exp/Cntr=0.3,0.1

Type RM Length L Ch R = 1 ,58      ,,,
XS GIS Cut Line= 6
2338615.48761906 577033.05140625  2338495.200987577503.346735572
2338512.43156988577701.4984386472338593.79821124 577822.11251878
2338916.39301287577637.3623801642339162.40744615577609.601996641
#Sta/Elev= 30
       0  2995.8    66.9 2988.19   102.3 2990.96   114.5 2988.51   163.5  2986.8
   253.2 2985.99   269.6 2980.84   310.4 2984.59   436.8 2984.28   453.2 2978.92
   469.5 2980.82   594.1 2982.45   623.62979.538   658.5 2978.43   664.92979.526
   678.6 2983.84   691.4    2985   786.6  2983.8   821.7 2984.51   832.5  2986.7
  1041.3 2985.47  1050.6 2982.03  1064.7 2985.51  1163.8 2987.02  1183.6 2982.83
  1195.2 2987.16  1204.2    2988  1401.1 2995.34  1425.1 3004.29  1455.4 3010.25
#Mann= 6 ,-1,0
       0     .06       0  160.62      .1       0   623.6    .045       0
   664.9      .1       0  942.47     .06       0 1326.51      .1       0
#XS Ineff= 2 , 0
          426.37 2988.02  908.62         2989.47
Permanent Ineff=
       F       F
Bank Sta=623.6,664.9
XS Rating Curve= 0 ,0
Exp/Cntr(USF)=0,0
Exp/Cntr=0.3,0.1
LCMann Table=0

Chan Stop Cuts=-1
Use User Specified Reach Order=0
Composite Channel Slope=5
